HEC-RAS study TROUTRN.prj: TROUTRN

--- TROUTRN.g01 (geometry) --- (continued)

Type RM Length L Ch R = 1 ,14615   ,262.2,263.5,265
XS GIS Cut Line= 4
2457845.47172407612861.5416594942457645.12275728613151.477562653
2457451.28920404613399.0632777112457356.81570751613509.825308131
#Sta/Elev= 30
       0 1972.08    45.4 1965.16   88.361962.012     201 1955.69   258.8 1949.68
     279 1948.19     342 1946.38  357.451946.651   419.2 1946.86     433 1943.61
   444.9 1939.59   458.4  1938.1   473.6 1940.16  500.161940.668   530.4 1941.96
   538.9 1941.19  556.031937.772   563.9 1935.72   575.9 1934.51  592.561937.771
   600.6 1940.15   610.8 1946.18   631.1 1960.48   654.8 1975.62   682.4 1994.47
   735.5 2028.02   747.8    2037   766.5 2048.86   787.6 2063.71   812.4 2080.16
#Mann= 6 ,-1 , 0
       0     .06       0   88.36     .05       0  357.45      .1       0
  500.16      .1       0  556.03    .045       0  592.56      .1       0
Bank Sta=556.03,592.56
XS Rating Curve= 0 ,0
Exp/Cntr(USF)=0,0
Exp/Cntr=0.3,0.1

Type RM Length L Ch R = 1 ,14352   ,230.6,237,238.4
XS GIS Cut Line= 4
2457674.10249452612759.0333799882457419.38468068613024.923027774
2457256.27590514613241.6566062212457173.60433398613328.796910958
#Sta/Elev= 30
       0  1966.7    27.5 1966.33   53.761962.227     189  1952.3   224.6 1948.62
   253.5 1943.67  315.651940.954   359.9 1939.16   375.8 1939.76   395.7 1937.13
   455.8 1938.91   465.8 1937.34  477.361932.579   482.4 1929.98     490 1929.56
   495.8 1929.95   502.3 1932.36   505.8 1934.35   510.8 1935.12   530.9 1934.53
   544.3  1932.6   561.5 1933.15   575.7 1930.54   580.9  1931.7     590 1939.59
   598.6 1949.74   621.4 1972.08     636 1983.36   663.2 2002.43   759.6  2061.9
#Mann= 5 ,-1 , 0
       0    .055       0   53.76     .05       0  315.65      .1       0
  477.36    .045       0   502.3      .1       0
Bank Sta=477.36,502.3
XS Rating Curve= 0 ,0
Exp/Cntr(USF)=0,0
Exp/Cntr=0.3,0.1

Type RM Length L Ch R = 1 ,14115   ,228,229,228.8
XS GIS Cut Line= 4
2457548.97795439612656.2525077352457318.83817521612852.876785089
2457106.57333034613056.2041628082457035.07359312 613136.64136718
#Sta/Elev= 30
       0  1965.5    10.2 1961.29   37.871961.595   41.171961.516   151.9 1948.33
     185  1948.5  223.581946.599   281.8 1940.97   315.5 1936.39   346.1 1935.05
   366.4 1934.93     375 1933.65   385.9 1930.94   391.5 1930.38   408.1 1929.67
   459.8 1930.54   496.7  1930.1   502.2 1929.78  508.991927.359   518.8 1925.21
   529.9 1924.49   536.2 1924.93  543.12 1927.36   552.1 1931.74   565.8 1943.26
   578.6 1953.13   600.2 1968.52   621.1 1981.35   640.9 1992.18   704.3  2029.3
#Mann= 6 ,-1 , 0
       0    .055       0   37.87     .06       0   41.17      .1       0
  223.58      .1       0  508.99    .045       0  543.12      .1       0
#XS Ineff= 2 , 0
          466.02 1930.38
Permanent Ineff=
       F       F
Bank Sta=508.99,543.12
XS Rating Curve= 0 ,0
Exp/Cntr(USF)=0,0
Exp/Cntr=0.3,0.1

Type RM Length L Ch R = 1 ,13886   ,231.9,258.8,277.6
XS GIS Cut Line= 4
2457350.11931024612511.0186665082457169.13560041612685.299275981
2456959.10512232612881.9235533352456883.13665153612953.423290555
#Sta/Elev= 30
       0 1965.44    19.3 1960.89    28.6 1954.84    32.4 1953.38    58.9 1953.09
   73.921951.336   126.7 1940.08  167.681935.841  194.731933.868   239.9 1929.71
   299.4 1929.86   306.3 1928.35   314.8 1924.55   320.3 1923.54   329.7 1924.23
   336.7 1923.56   347.5 1924.98     356 1925.03     386 1923.29   406.9 1925.48
  434.591926.215   452.2 1924.72   462.7 1920.94     472 1920.64   480.5 1921.15
  486.971924.332   499.4 1931.59  512.251940.438   550.4 1964.53   643.3  2016.9
#Mann= 8 ,-1 , 0
       0    .055       0   73.92     .06       0  167.68      .1       0
  194.73      .1       0  434.59      .1       0   452.2    .045       0
  486.97      .1       0  512.25      .1       0
#XS Ineff= 2 , 0
          434.24 1928.24
Permanent Ineff=
       F       F
Bank Sta=452.2,486.97
XS Rating Curve= 0 ,0
Exp/Cntr(USF)=0,0
Exp/Cntr=0.5,0.3

Type RM Length L Ch R = 1 ,13627   ,101.7,95.2,84.5
XS GIS Cut Line= 4
2457212.73133426612471.6509270582456998.99319262612616.992863376
2456926.32222446612590.2755956712456767.08730894 612770.88432536
#Sta/Elev= 30
       0 1948.83    16.9 1948.69    26.8 1947.81    48.4 1940.06    65.3 1935.86
    99.1 1930.55  137.261927.354   181.4 1926.05   196.7 1924.75   216.8 1921.68
   231.2 1921.27  253.121921.705   267.3 1921.75   279.21920.476   288.3 1918.86
   297.1 1918.14   309.9 1918.02   318.4  1918.4  325.691920.477     332 1921.76
   344.5 1922.21   395.6  1921.3   413.9 1921.31   443.4 1922.21   449.4 1923.32
   455.1 1925.26  465.831930.463  499.351949.424   540.1 1971.27   576.7 1990.22
#Mann= 7 ,-1 , 0
       0    .055       0  137.26      .1       0  253.12      .1       0
   279.2    .045       0  325.69      .1       0  465.83      .1       0
  499.35      .1       0
#XS Ineff= 2 , 0
             255  1921.3     348          1921.3
Permanent Ineff=
       F       F
Bank Sta=279.2,325.69
XS Rating Curve= 0 ,0
Exp/Cntr(USF)=0,0
Exp/Cntr=0.5,0.3

Type RM Length L Ch R = 1 ,13532   ,125.1,115.6,94.8
XS GIS Cut Line= 4
2457097.31273778612400.0486496082457013.95486254612509.055101846
2456938.07782225612513.329864679 2456748.9195669612730.274078447
#Sta/Elev= 30
       0 1944.02    15.3 1944.16    23.8 1943.72   37.991940.922   71.971934.771
   109.3 1927.75   144.4 1925.99   148.5 1924.85  158.061918.801   160.5 1917.55
   164.5  1916.5   172.5 1916.06   196.5 1918.55   200.5 1918.66   212.6 1917.72
   230.5 1917.39   236.6 1918.35   241.8 1919.91   247.9 1920.94  279.421920.989
   300.2 1920.94   326.7 1919.89   344.3 1916.86   378.3  1921.4   390.4 1921.48
   395.3  1922.2     401 1924.34   411.7 1929.77   464.7 1961.14   501.1 1980.04
#Mann= 6 ,-1 , 0
       0    .055       0   37.99     .06       0   71.97      .1       0
  158.06    .045       0   196.5      .1       0  279.42      .1       0
#XS Ineff= 2 , 0
                          258.87         1921.35
Permanent Ineff=
       F       F
Bank Sta=158.06,196.5
XS Rating Curve= 0 ,0
Exp/Cntr(USF)=0,0
Exp/Cntr=0.5,0.3

Type RM Length L Ch R = 1 ,13416   ,181.4,184,181.6
XS GIS Cut Line= 4
2456995.67130902612336.1619248882456971.23850819612373.625552824
2456746.45674057612630.9843882132456687.81801859612709.169350863
#Sta/Elev= 30
       0 1940.12    25.8 1939.83    34.4 1938.31   41.651935.429    46.4 1933.24
   53.441931.665    63.7 1929.34    67.7 1926.36   77.33 1916.78      82 1913.89
    85.7  1913.3    99.5 1915.04   106.3 1914.49     114 1916.36     142 1916.96
   153.7 1915.36   167.9 1917.65  192.781917.176   209.7 1914.82     227 1918.46
   252.9  1918.3   281.3 1917.16   315.3 1919.53   338.5 1918.46   349.3 1919.29
   359.8 1923.48   386.4 1939.47   405.9 1950.33   461.3 1978.78   484.2 1989.66
#Mann= 6 ,-1 , 0
       0    .055       0   41.65     .06       0   53.44      .1       0
   77.33    .045       0     114      .1       0  192.78      .1       0
#XS Ineff= 2 , 0
                          318.55         1919.72
Permanent Ineff=
       F       F
Bank Sta=77.33,114
XS Rating Curve= 0 ,0
Exp/Cntr(USF)=0,0
Exp/Cntr=0.3,0.1

Type RM Length L Ch R = 1 ,13232   ,156.6,168.3,162.8
XS GIS Cut Line= 4
2456876.76501166612213.9979207472456788.80692868612336.161924888
2456673.15833809612552.7994255632456616.14846949612630.984388213
#Sta/Elev= 30
       0 1942.08      25 1939.81    36.5 1934.48   54.221935.087    92.5 1933.61
  101.671930.338   106.1 1928.73   113.8 1927.17   145.4 1922.39   158.2    1921
   162.7 1919.82   171.8 1915.21   176.3 1913.65  187.761913.191     199 1910.94
   213.2 1910.25   221.6 1910.57  243.521913.191   251.6 1914.12   285.1 1914.97
   312.3 1914.53   325.9 1916.19     3511916.053   358.1 1916.42   367.3 1919.61
   393.9 1931.92   431.2 1947.12   458.1 1959.63   487.8 1974.43   492.9 1976.42
#Mann= 6 ,-1 , 0
       0    .055       0   54.22     .06       0  101.67      .1       0
  187.76    .045       0  243.52      .1       0     351      .1       0
#XS Ineff= 2 , 0
                          343.41          1916.3
Permanent Ineff=
       F       F
Bank Sta=187.76,243.52
XS Rating Curve= 0 ,0
Exp/Cntr(USF)=0,0
Exp/Cntr=0.3,0.1

Type RM Length L Ch R = 1 ,13064   ,110.7,110.4,112.7
XS GIS Cut Line= 4
2456749.71444735612116.2667174352456692.70457875612228.657601244
2456577.05598817612427.3777146462456511.90185262612547.912865398
#Sta/Elev= 30
       0  1946.3    34.3 1939.56    39.9 1937.61   47.281933.074    52.3 1930.37
    56.8 1929.84    87.5  1930.3    97.1 1931.43  112.04 1930.69   119.6 1927.81
   137.9  1914.5   140.8 1913.25   162.11909.573   165.6 1907.24   170.3 1905.96
   205.2 1909.56   237.5 1910.95     249 1909.66   272.4 1908.66     286 1910.77
   299.8 1909.93   304.5 1910.92   313.7 1915.39   318.4 1916.65  366.211917.648
     378 1919.36   389.8 1922.51   419.3 1933.51   460.6 1951.85     493 1967.95
#Mann= 6 ,-1 , 0
       0    .055       0   47.28     .06       0  112.04      .1       0
   162.1    .045       0   205.2      .1       0  366.21      .1       0
Bank Sta=162.1,205.2
XS Rating Curve= 0 ,0
Exp/Cntr(USF)=0,0
Exp/Cntr=0.3,0.1

Type RM Length L Ch R = 1 ,12954   ,173.9,174.1,174.7
XS GIS Cut Line= 4
2456666.64292454612055.9991420592456599.85993561612168.390025868
2456477.69593147612385.0275265442456420.68606287612469.727902748
#Sta/Elev= 30
       0 1948.08      39 1941.07    60.4 1926.64   85.24 1926.89   85.411926.886
    95.4 1926.69   105.7 1928.63     115 1928.66   133.6 1924.97   142.2  1922.2
     152 1917.06   156.6 1914.03   164.61906.414   170.3 1903.35   179.5 1903.02
   184.1 1903.34   192.1 1905.94   200.9 1907.31   214.4 1907.51   234.6 1906.25
   248.4 1908.51   262.6 1909.11   312.7 1908.96   326.5 1907.54  334.44 1908.92
   349.4  1914.7     377 1915.87   391.6 1920.31   429.9 1936.66   481.5 1962.57
#Mann= 6 ,-1 , 0
       0    .055       0   85.24     .06       0   85.41      .1       0
   164.6    .045       0   192.1      .1       0  334.44      .1       0
Bank Sta=164.6,192.1
XS Rating Curve= 0 ,0
Exp/Cntr(USF)=0,0
Exp/Cntr=0.3,0.1

Type RM Length L Ch R = 1 ,12779   ,298.4,302.6,298.9
XS GIS Cut Line= 4
2456546.10777378611950.1236718042456476.06707808612051.112581894
2456350.64536716612248.2038419072456269.20269773612362.223579104
#Sta/Elev= 30
       0 1951.69    12.9 1946.47    25.3 1942.74      74  1931.2    86.3 1923.17
    89.2 1921.79   112.9  1921.7  125.93 1920.46   132.4 1919.26   136.9 1917.21
  153.711903.483   155.8 1902.03   160.6 1900.37     170 1899.69   175.9 1900.54
   184.3 1903.99   201.9 1904.66   217.5 1902.47   239.6 1903.55   254.1  1905.1
   307.5 1904.16   312.3 1904.56   321.8 1907.09     334 1907.42  370.841912.108
     377 1913.56   390.8 1918.29   404.1  1924.1   435.8 1939.99   496.6 1973.12
#Mann= 5 ,-1 , 0
       0    .055       0  125.93      .1       0  153.71    .045       0
   184.3      .1       0  370.84      .1       0
Bank Sta=153.71,184.3
XS Rating Curve= 0 ,0
Exp/Cntr(USF)=0,0
Exp/Cntr=0.3,0.1

Type RM Length L Ch R = 1 ,12477   ,117.7,116.9,112.7
XS GIS Cut Line= 4
2456335.98568666611845.8770549382456277.34696468611941.979404862
2456221.96594947612064.143409002 2456132.3790131612227.028747856
#Sta/Elev= 30
       0 1926.05    19.1 1922.36    48.5  1914.3    56.9 1913.56    74.4 1914.64
    92.21914.083     109 1912.13   122.4 1907.33   133.4 1905.69   135.5  1904.9
   144.3 1898.66   148.5 1897.64  164.071899.237   175.1 1898.73   183.8 1899.31
   193.8 1898.58   208.9  1901.4   232.2 1901.72   251.1 1900.67  265.931898.309
  285.871895.247     313 1891.32   319.51895.245   322.9 1898.24     332 1908.69
   341.1 1917.23   351.2    1925     363 1932.93   382.2 1943.65   432.6 1968.69
#Mann= 6 ,-1 , 0
       0    .055       0    92.2     .06       0  164.07      .1       0
  265.93      .1       0  285.87    .045       0   319.5      .1       0
#XS Ineff= 2 , 0
          222.45 1901.97
Permanent Ineff=
       F       F
Bank Sta=285.87,319.5
XS Rating Curve= 0 ,0
Exp/Cntr(USF)=0,0
Exp/Cntr=0.3,0.1

Type RM Length L Ch R = 1 ,12360   ,176.1,175.7,174.8
XS GIS Cut Line= 4
2456215.45053591611790.4960397282456164.95608087611904.515776925
2456085.14226483612090.2050632192456042.79207673612176.534292811
#Sta/Elev= 30
       0 1916.02      19  1913.4    52.4 1911.07    74.8 1911.18   90.111910.421
     107  1908.8   118.5 1906.19  124.481905.585   144.7 1905.28   152.6 1903.96
   162.1 1897.23   166.5 1895.34   170.8 1894.72   188.2 1896.02   192.6 1895.14
   196.9 1895.06     210 1896.29   231.7 1895.41   239.6 1894.51  253.641892.754
   262.3 1890.18   271.3 1889.81   283.5 1890.23  293.981892.754   301.8 1895.69
     332 1917.41   363.2  1936.7   400.9 1957.23   416.7  1966.7     423 1971.06
#Mann= 6 ,-1 , 0
       0    .055       0   90.11     .06       0  124.48      .1       0
   239.6      .1       0  253.64    .045       0  293.98      .1       0
#XS Ineff= 2 , 0
          211.54 1898.78
Permanent Ineff=
       F       F
Bank Sta=253.64,293.98
XS Rating Curve= 0 ,0
Exp/Cntr(USF)=0,0
Exp/Cntr=0.3,0.1

Type RM Length L Ch R = 1 ,12184   ,150.5,151.5,151.7
XS GIS Cut Line= 4
2456042.79207673611709.0533703012455971.12252763611907.773483702
2455923.88577936612026.6797810662455886.42215143612106.493597104
#Sta/Elev= 30
       0 1915.88   18.971915.284    31.7 1915.08    44.5 1913.95    70.2 1909.02
    78.5 1907.98   116.8 1906.89     121 1906.14   125.3 1904.58  130.121901.151
   133.8 1898.37     138 1896.17   142.3 1895.23   186.31893.888   193.3 1894.21
   206.1  1893.2     249    1894     254 1893.46  274.631888.302   283.5 1885.48
     294 1884.84   296.4 1884.92   300.7 1886.16  303.64  1888.3   317.9 1900.51
   327.9 1908.11   365.9 1933.09   379.2 1941.18   401.3 1956.52   427.4 1973.31
#Mann= 6 ,-1 , 0
       0      .1       0   18.97    .055       0  130.12     .06       0
   186.3      .1       0  274.63    .045       0  303.64      .1       0
#XS Ineff= 2 , 0
          245.97 1894.19
Permanent Ineff=
       F       F
Bank Sta=274.63,303.64
XS Rating Curve= 0 ,0
Exp/Cntr(USF)=0,0
Exp/Cntr=0.3,0.1

Type RM Length L Ch R = 1 ,12033   ,184.6,185.4,183.6
XS GIS Cut Line= 4
2455928.77233953611666.7031821992455840.81425655611845.877054938
2455796.83521506611940.3505514732455749.59846679612034.824048008
#Sta/Elev= 30
       0 1914.03    58.1 1909.05    80.4 1906.48   102.7 1906.21   121.2 1905.08
   129.4 1904.06   133.2 1903.03   138.3 1900.02   142.1 1898.39  145.13 1897.58
   149.8 1896.76   205.1 1891.29     223 1888.44     236 1887.29  240.991885.184
   244.8 1882.89   247.1 1882.47   262.5 1881.78   268.2 1882.47   271.2 1883.58
     273 1885.19   275.7 1887.81   280.1 1892.67   284.5  1894.7   306.6 1895.76
   311.1 1897.18   313.8  1898.6   340.1 1914.04   362.1 1928.79   409.4 1957.36
#Mann= 4 ,-1 , 0
       0    .055       0  145.13      .1       0  240.99    .045       0
     273      .1       0
Bank Sta=240.99,273
XS Rating Curve= 0 ,0
Exp/Cntr(USF)=0,0
Exp/Cntr=0.3,0.1

Type RM Length L Ch R = 1 ,11847   ,269.2,262.5,256.1
XS GIS Cut Line= 4
 2455733.3099329611639.0126745942455700.73286513611723.713050797
2455660.01153042611824.7019608872455622.54790248611964.783352301
#Sta/Elev= 30
       0 1919.75    25.6 1912.31   41.311904.888    45.2 1903.22    48.3  1902.5
      77  1900.4    85.6 1901.61    89.9 1900.87   102.8 1896.74   107.4 1894.53
   120.1 1886.58   130.41881.431   137.3 1878.71   141.6 1878.21   154.6 1878.67
   158.9 1880.08     1611881.429   165.4 1883.96   171.8 1886.21   184.7 1889.19
   189.1 1889.48   214.3 1887.71     235 1885.41   239.2 1885.52   243.3 1886.27
   254.7 1891.25   268.8 1898.92   301.3 1914.28   330.3 1929.36   344.6  1937.5
#Mann= 4 ,-1 , 0
       0      .1       0   41.31     .06       0   130.4    .045       0
     161      .1       0
#XS Ineff= 2 , 0
                          190.05         1889.26
Permanent Ineff=
       F       F
Bank Sta=130.4,161
XS Rating Curve= 0 ,0
Exp/Cntr(USF)=0,0
Exp/Cntr=0.3,0.1

Type RM Length L Ch R = 1 ,11585   ,197.1,195.2,194.2
XS GIS Cut Line= 4
2455440.11632297611518.4775238422455425.45664247611658.558915256
 2455435.2297628611779.0940660082455454.77600346611930.577431142
#Sta/Elev= 30
       0 1949.81    5.04 1947.57    93.3 1910.08    96.9  1908.3  105.921900.453
     109 1898.62   121.1 1895.02   133.1 1889.77   144.2 1889.73   177.3 1886.08
   181.3 1884.02   185.3 1880.66   189.3 1876.41   192.21874.387   197.4 1871.91
   209.4 1870.65   217.4 1871.38  222.731874.388   229.5 1879.16   237.5 1879.35
   245.5 1880.23   257.7 1880.44   269.6 1879.91   297.9 1880.86     314 1879.53
     318 1880.18   326.1 1884.56   354.3  1903.8   394.7 1925.29   414.5 1937.26
#Mann= 5 ,-1 , 0
       0      .1       0    5.04      .1       0  105.92     .06       0
   192.2    .045       0  222.73      .1       0
Bank Sta=192.2,222.73
XS Rating Curve= 0 ,0
Exp/Cntr(USF)=0,0
Exp/Cntr=0.3,0.1

Type RM Length L Ch R = 1 ,11390   ,182.7,179.5,176.2
XS GIS Cut Line= 4
2455177.87092741611521.7352306192455229.99423585611704.166810135
2455254.42703667611850.7636151032455275.60213072611945.237111639
#Sta/Elev= 30
       0  1989.7    30.3 1971.01    38.6 1964.04    51.1  1960.2    55.3 1957.55
    71.9 1942.36    80.2 1936.01   117.7 1912.16  140.511899.268   146.8 1894.22
   155.1 1884.62   159.3  1882.5   180.1 1881.18   212.8 1876.08     233 1877.17
  238.431875.747  246.191870.792   251.8 1867.93   257.4 1867.39   265.5 1867.55
   269.5 1868.58  273.02 1870.79   277.7 1873.76   281.7 1874.84     302 1873.99
   310.1 1875.74   338.4 1892.11   353.9 1904.49   372.2 1916.54   435.2 1946.89
#Mann= 5 ,-1 , 0
       0      .1       0  140.51     .06       0  238.43      .1       0
  246.19    .045       0  273.02      .1       0
#XS Ineff= 2 , 0
          231.18  1877.2  288.46         1877.95
Permanent Ineff=
       F       F
Bank Sta=246.19,273.02
XS Rating Curve= 0 ,0
Exp/Cntr(USF)=0,0
Exp/Cntr=0.3,0.1

Type RM Length L Ch R = 1 ,11210   ,128.5,123.5,120.2
XS GIS Cut Line= 4
2454987.29508095611650.4146483132455044.30494955611766.063238899
2455091.54169782611873.5675625432455153.43812658611972.927619244
#Sta/Elev= 30
       0 1933.01   43.521918.197    58.5 1913.01    94.2 1898.58    98.6 1896.03
   116.4 1879.23   119.4 1877.81   122.4 1877.18   138.6 1876.94   160.4 1874.22
  170.671873.752   176.9 1872.11  183.651867.181   186.6 1865.41     191 1864.12
   199.7 1863.91   207.3 1864.79  212.021867.183   221.6 1873.89   252.4 1886.91
     270 1895.77   272.9    1898   276.2 1901.64   280.9 1907.98   285.6 1913.13
   290.3 1915.73   299.8 1919.68   319.3 1925.92   342.2 1932.68   363.4 1937.38
#Mann= 5 ,-1 , 0
       0      .1       0   43.52     .06       0  170.67      .1       0
  183.65    .045       0  212.02      .1       0
Bank Sta=183.65,212.02
XS Rating Curve= 0 ,0
Exp/Cntr(USF)=0,0
Exp/Cntr=0.3,0.1

Type RM Length L Ch R = 1 ,11087   ,135.1,129.2,125.1
XS GIS Cut Line= 4
 2454824.4097421611767.6920922882454940.05833269  611865.4232956
2455019.87214872 611955.010231972455089.91284443611995.731566683
#Sta/Elev= 30
       0 1971.02     8.3  1965.4    18.8  1959.9      45 1944.36    63.81931.494
    76.4 1922.72    86.8 1920.12   100.4 1911.11   120.3 1899.21   123.5 1896.79
     134  1885.8   140.2  1877.9     143 1876.15   167.5 1873.83     194 1870.12
   196.9 1869.41  206.021864.273   213.9  1861.9     223 1860.97   230.9 1861.49
   233.6 1862.11  237.581864.275   250.7 1875.01   257.7 1879.57     291 1891.76
   307.1 1900.69   316.4  1908.5   320.2 1910.87   330.2  1915.7   352.4 1923.58
#Mann= 4 ,-1 , 0
       0      .1       0    63.8     .06       0  206.02    .045       0
  237.58      .1       0
Bank Sta=206.02,237.58
XS Rating Curve= 0 ,0
Exp/Cntr(USF)=0,0
Exp/Cntr=0.3,0.1

Type RM Length L Ch R = 1 ,10957   ,152,150.9,146.9
XS GIS Cut Line= 4
2454755.99789978611933.8351379192454861.87337004611995.731566683
2454979.15081401612060.8857022252455063.85119021612108.122450492
#Sta/Elev= 30
       0 1961.55      31  1939.6    49.5  1925.3    58.8 1919.32      68 1911.45
    72.7 1909.65    77.3 1908.76    81.7 1906.73    91.2 1899.72   114.4 1884.83
   132.8 1870.74   137.3 1869.38  142.421869.756   152.1  1869.7   178.5    1867
  187.251861.315   192.3 1858.83   199.1 1857.98   215.2 1859.26   219.7 1860.16
  221.731861.317   228.6  1866.2   237.4  1871.2   252.1 1881.62   256.3 1884.09
   277.3 1893.33  285.671896.616   297.6 1900.88   320.5 1910.33   353.8 1925.29
#Mann= 5 ,-1 , 0
       0      .1       0  142.42     .06       0  187.25    .045       0
  221.73     .06       0  285.67      .1       0
Bank Sta=187.25,221.73
XS Rating Curve= 0 ,0
Exp/Cntr(USF)=0,0
Exp/Cntr=0.3,0.1

Type RM Length L Ch R = 1 ,10806   ,173,176.2,175.3
XS GIS Cut Line= 4
2454692.47261763612091.8339166072454842.32712937612160.245758926
2454961.23342674612205.8536538052455047.56265633612244.946135129
#Sta/Elev= 30
       0 1954.81    28.9 1932.44    37.7 1925.85    46.5 1920.17    55.3 1913.25
    67.4  1905.3   74.031902.894    94.8 1889.36   112.4  1879.8     130 1868.72
   138.8 1864.55   143.2 1864.22   160.8 1865.41     178 1864.59   182.6 1863.53
   190.9  1858.7   195.2 1856.39   203.7 1855.35   220.9 1856.19  226.931858.699
   229.4 1860.07   233.7 1860.95   242.3 1860.67  250.681861.231   255.1 1862.58
   259.4 1864.92   275.5 1876.37   298.1  1889.2   324.5 1901.24   386.9 1931.73
#Mann= 5 ,-1 , 0
       0      .1       0   74.03     .06       0   190.9    .045       0
  226.93     .06       0  250.68      .1       0
Bank Sta=190.9,226.93
XS Rating Curve= 0 ,0
Exp/Cntr(USF)=0,0
Exp/Cntr=0.3,0.1

Type RM Length L Ch R = 1 ,10630   ,186,190.3,192.5
XS GIS Cut Line= 4
 2454625.6896287612249.8326952952454762.51331333 612311.72912406
2454904.22355814612368.7389926582455018.24329534612401.316060429
#Sta/Elev= 30
       0 1951.28    31.7 1931.19    49.5 1921.01      59 1914.46    71.4  1909.3
    80.2 1903.72  124.591878.629   137.3 1871.26   150.4 1861.72   154.7 1860.01
   180.6 1861.97   189.2  1861.9   210.8  1858.2  219.081855.537   223.7 1854.24
   249.6 1852.37  263.151855.538   271.1 1856.69   275.5 1858.21   279.8  1860.5
   284.1 1864.74   288.4 1871.46   292.7 1876.72     297 1880.78   305.5 1887.46
  354.351915.119   368.2 1922.23   405.4 1945.42   417.9 1950.79   421.5 1952.89
#Mann= 5 ,-1 , 0
       0      .1       0  124.59     .06       0  219.08    .045       0
  263.15      .1       0  354.35      .1       0
#XS Ineff= 2 , 0
          184.81 1862.63
Permanent Ineff=
       F       F
Bank Sta=219.08,263.15
XS Rating Curve= 0 ,0
Exp/Cntr(USF)=0,0
Exp/Cntr=0.3,0.1

Type RM Length L Ch R = 1 ,10440   ,165.3,168.6,171.1
XS GIS Cut Line= 4
2454537.73154572612368.7389926582454726.67853879612486.016436633
2454817.89432854 612544.655158622454920.51209202612609.809294162
#Sta/Elev= 30
       0 1952.91    34.4  1934.4      53 1925.22    66.2 1916.61    76.5 1913.86
    90.6 1904.53   104.8 1896.79  128.071885.387   161.3 1868.98   173.7 1859.66
   180.1  1855.8   184.8 1855.29     213 1858.09   231.7 1855.37   246.2 1856.37
   253.6 1854.91  261.441851.181   269.4 1848.51   275.2 1847.91     289 1849.01
  294.27 1851.18   322.3 1870.93   327.1 1874.99   331.8 1879.91   336.6 1883.65
   372.3 1904.51   398.2 1921.93   411.91933.287  424.371941.018   452.4 1959.66
#Mann= 6 ,-1 , 0
       0      .1       0  128.07     .06       0  261.44    .045       0
  294.27      .1       0   411.9      .1       0  424.37     .12       0
#XS Ineff= 2 , 0
           245.3 1856.82
Permanent Ineff=
       F       F
Bank Sta=261.44,294.27
XS Rating Curve= 0 ,0
Exp/Cntr(USF)=0,0
Exp/Cntr=0.3,0.1

Type RM Length L Ch R = 1 ,10271   ,170.7,170.6,170.5
XS GIS Cut Line= 4
2454490.49479745612481.1298764672454633.83389564612609.809294162
2454716.90541846  612689.62311022454808.12120821 612767.80807285
#Sta/Elev= 30
       0 1932.97    12.8 1926.28    21.8  1919.5    35.4 1915.85    46.7 1908.27
    54.1 1904.15    70.2 1896.12   99.651883.171   129.3 1869.95   150.8 1854.39
   154.4 1852.64   157.2  1852.2   182.7 1854.36   188.5 1854.01   199.7 1850.65
     211 1851.96  224.74 1850.75   228.8 1849.59  234.521845.336   239.3 1842.26
   251.9  1841.6   259.1 1842.84  263.36 1845.34   269.2 1851.65  282.641862.362
     293 1869.71   326.1  1888.6   352.6 1901.37   383.8 1917.56     428 1942.23
#Mann= 6 ,-1 , 0
       0      .1       0   99.65     .06       0  224.74      .1       0
  234.52    .045       0  263.36      .1       0  282.64      .1       0
Bank Sta=234.52,263.36
XS Rating Curve= 0 ,0
Exp/Cntr(USF)=0,0
Exp/Cntr=0.3,0.1

Type RM Length L Ch R = 1 ,10101   ,222.7,218.7,214.9
XS GIS Cut Line= 4
2454379.73276703612632.6132416012454493.75250423 612712.42705764
2454588.22600076612802.0139940092454677.81293713612891.600930379
#Sta/Elev= 30
       0 1923.59     6.7 1919.58    15.3 1916.84    29.6 1908.13    52.6  1895.6
   60.661891.915    72.7 1884.69    81.3 1876.81   108.6 1855.89   118.7 1850.51
   122.5 1849.55   135.5 1850.46   157.1 1850.32   164.3 1849.09   172.7 1845.35
   177.6  1844.3  193.731844.135   200.9 1843.67  206.511842.255   217.7 1839.08
   220.8 1838.87   232.2 1839.67     235 1840.71  236.931842.257   247.4 1852.07
   264.8 1862.54  316.041880.838  321.631882.825   359.5 1898.54   396.1 1915.93
#Mann= 7 ,-1 , 0
       0      .1       0   60.66     .06       0  193.73      .1       0
  206.51    .045       0  236.93      .1       0  316.04     .12       0
  321.63      .1       0
Bank Sta=206.51,236.93
XS Rating Curve= 0 ,0
Exp/Cntr(USF)=0,0
Exp/Cntr=0.3,0.1

Type RM Length L Ch R = 1 ,9882    ,184.2,175.8,168.4
XS GIS Cut Line= 4
2454221.73398834612780.8388999582454321.09404504612875.312396494
2454453.03116951612946.9819455892454570.30861349612997.476400634
#Sta/Elev= 30
       0 1943.07    14.6 1930.74    26.2 1923.58    53.1 1905.17    64.4 1900.17
    78.4 1890.99    89.9 1884.76     121 1869.44   126.7 1864.88   135.1 1853.69
     138 1850.93   143.5 1848.54  147.261848.633   175.4 1844.65   189.1 1843.51
  201.171837.625   207.3  1834.6   214.7  1834.2   225.5 1835.28  231.441837.627
   241.3 1839.63   248.2 1842.57  272.811842.605   288.5 1842.27   294.6 1842.89
   297.6 1843.85  311.141852.102   328.9 1858.41  391.471876.875   414.9 1885.21
#Mann= 7 ,-1 , 0
       0      .1       0  147.26     .06       0  201.17    .045       0
  231.44     .06       0  272.81      .1       0  311.14      .1       0
  391.47     .12       0
#XS Ineff= 2 , 0
                          252.02         1843.01
Permanent Ineff=
       F       F
Bank Sta=201.17,231.44
XS Rating Curve= 0 ,0
Exp/Cntr(USF)=0,0
Exp/Cntr=0.3,0.1

Type RM Length L Ch R = 1 ,9706    ,239.7,226,213.9
XS GIS Cut Line= 4
2454143.54902569613039.8265887362454304.80551116613083.805630226
 2454469.3197034613080.5479234492454581.71058721613061.001682787
#Sta/Elev= 30
       0 1895.01    15.8  1887.8      24  1882.8    36.5 1878.73    57.2 1866.61
    77.9 1857.32    86.2 1851.77    94.5  1847.6   106.1 1844.37  121.18 1844.19
     136 1843.98   160.9  1839.9   185.1 1839.91   189.1 1838.88   197.1 1835.06
  203.631833.706   217.1  1830.5   225.1 1829.87   229.1 1830.31  235.991833.704
   245.1 1838.39   269.1 1837.03   277.1 1837.96   297.1  1837.7   309.1 1839.17
   329.1 1839.46   333.1 1840.32   365.6 1855.54  424.891879.007   445.8 1887.32
#Mann= 5 ,-1 , 0
       0      .1       0  121.18     .06       0  203.63    .045       0
  235.99      .1       0  424.89     .12       0
Bank Sta=203.63,235.99
XS Rating Curve= 0 ,0
Exp/Cntr(USF)=0,0
Exp/Cntr=0.3,0.1

Type RM Length L Ch R = 1 ,9480    ,197.5,194.9,192.6
XS GIS Cut Line= 4
 2454298.2900976  613414.46286812454428.59836869613310.216251233
2454545.87581266613194.5676606472454627.31848209613114.753844609
#Sta/Elev= 30
       0 1853.19     5.7 1848.12      16  1840.7    19.9 1838.72    24.9  1837.3
    41.6 1837.04    51.8 1836.19   71.081836.048   105.3 1836.33   133.8 1832.31
   159.4 1832.69   175.5 1831.96   196.2 1832.86   200.1 1832.18  205.421829.923
   210.3 1828.32     216 1828.18   224.5 1826.43   228.6 1826.17   235.8 1826.76
  246.391829.922  252.211831.265  253.761831.389     271 1832.29   287.9 1834.97
   293.5  1837.1   309.3 1845.17  375.491871.235   422.6 1890.18   445.6 1900.16
#Mann= 7 ,-1 , 0
       0      .1       0   71.08     .06       0  205.42    .045       0
  246.39     .06       0  252.21      .1       0  253.76      .1       0
  375.49     .12       0
#XS Ineff= 2 , 0
          192.93 1835.94
Permanent Ineff=
       F       F
Bank Sta=205.42,246.39
XS Rating Curve= 0 ,0
Exp/Cntr(USF)=0,0
Exp/Cntr=0.3,0.1

Type RM Length L Ch R = 1 ,9285    ,232,236.6,243.8
XS GIS Cut Line= 4
2454479.09282373613549.6576993482454570.30861349613456.813056202
2454669.66867019613331.3913452842454772.28643367 613191.30995387
#Sta/Elev= 30
       0 1913.46    18.7 1909.34    27.2 1906.14    31.9 1902.18    39.5 1893.28
    48.7 1876.25    52.6 1871.17   73.591854.427    85.1 1846.49    96.5 1837.27
   104.8  1831.8   109.2 1829.98   147.9 1829.89   168.3 1827.98   185.9 1829.82
   188.8  1829.5  194.461826.501   201.7 1824.13   214.3 1824.07   224.5 1822.84
   234.3 1823.59  240.24  1826.5   244.9 1828.77   254.3 1830.91   270.4 1838.08
   295.7 1852.31  304.71  1856.6   325.5 1866.53   362.8 1886.88   463.8 1938.71
#Mann= 5 ,-1 , 0
       0      .1       0   73.59     .06       0  194.46    .045       0
  240.24      .1       0  304.71      .1       0
#XS Ineff= 2 , 0
          183.62 1831.73
Permanent Ineff=
       F       F
Bank Sta=194.46,240.24
XS Rating Curve= 0 ,0
Exp/Cntr(USF)=0,0
Exp/Cntr=0.3,0.1

Type RM Length L Ch R = 1 ,9049    ,192.2,200.2,208.4
XS GIS Cut Line= 4
2454614.28765498613650.6466094382454755.99789978613577.348206953
2454917.25438525 613469.843883312455078.51087071613406.318601157
#Sta/Elev= 30
       0 1920.96     9.1 1921.52      14 1918.49      23 1905.22    29.8 1897.99
    44.7  1885.9    63.6 1872.58    72.6  1864.6   77.59 1857.66    81.6 1852.62
    99.6 1836.44     104 1830.92   112.9 1824.62   117.6 1822.74   131.1 1822.48
   177.7 1829.18   185.6 1827.38   192.1 1822.94   200.8    1819   215.7  1818.7
   221.7 1819.09  228.511822.037  256.631842.994   268.6 1850.07   286.6 1855.31
   311.9 1864.78   363.6 1892.17   427.7 1932.08   506.8 1983.21   526.7  1998.4
#Mann= 5 ,-1 , 0
       0      .1       0   77.59     .06       0   192.1    .045       0
  228.51     .06       0  256.63      .1       0
#XS Ineff= 2 , 0
          175.81 1828.37
Permanent Ineff=
       F       F
Bank Sta=192.1,228.51
XS Rating Curve= 0 ,0
Exp/Cntr(USF)=0,0
Exp/Cntr=0.3,0.1

Type RM Length L Ch R = 1 ,8849    ,181.6,199.9,215
XS GIS Cut Line= 4
2454643.60701597613733.7181322532454783.68840739 613748.37781275
2454961.23342674613719.0584517562455159.95354014613671.821703488
#Sta/Elev= 30
       0 1897.31     7.2 1896.22    20.2 1892.45    23.3 1891.24   26.62 1888.52
    35.3 1880.14    47.4 1871.37      84 1848.54   111.7 1834.25   127.8 1821.17
   131.9 1820.66   156.1 1824.81   168.3  1825.7   172.3 1825.47   184.5 1821.17
  211.18 1817.83   229.1 1814.89   241.2 1814.55   245.3 1814.86  251.29 1817.83
   261.5 1822.62   273.9  1830.2   318.8 1863.06   359.4 1889.39     372 1898.51
   412.8 1922.79     458 1951.88   466.3 1958.26     475 1966.23   525.1 2000.87
#Mann= 4 ,-1 , 0
       0      .1       0   26.62     .06       0  211.18    .045       0
  251.29      .1       0
#XS Ineff= 2 , 0
          164.52 1825.52
Permanent Ineff=
       F       F
Bank Sta=211.18,251.29
XS Rating Curve= 0 ,0
Exp/Cntr(USF)=0,0
Exp/Cntr=0.3,0.1

Type RM Length L Ch R = 1 ,8649    ,163.9,179.4,193.2
XS GIS Cut Line= 4
2454646.86472275613782.5837339092454762.51331334613849.366722839
2454910.73897169613973.159580368  2455037.789536614088.808170954
#Sta/Elev= 30
       0 1871.17   39.111860.592    55.3 1855.01    59.9 1852.83    64.5 1849.33
    87.6 1820.97    93.8 1816.96    96.9 1816.57   133.8 1822.33   139.1 1821.42
   149.5 1817.41  173.461819.224   185.9 1816.65     217 1815.03  224.261810.854
   229.5 1808.45   239.9 1807.94   253.7 1808.45  262.681810.853   269.3  1812.8
   276.8 1816.91   300.6 1837.63   313.7 1846.68   388.7 1890.83   441.2 1924.08
   445.7  1927.6   449.7 1933.26     461 1956.97   466.6 1964.95   498.5 1986.95
#Mann= 5 ,-1 , 0
       0      .1       0   39.11     .06       0  173.46      .1       0
  224.26    .045       0  262.68      .1       0
Bank Sta=224.26,262.68
XS Rating Curve= 0 ,0
Exp/Cntr(USF)=0,0
Exp/Cntr=0.3,0.1

Type RM Length L Ch R = 1 ,8469    ,117,120.6,123.4
XS GIS Cut Line= 4
2454638.72045581613800.5011211832454671.29752358 613893.34576433
2454687.58605746614049.7156896292454689.21491085614224.003002203
#Sta/Elev= 30
       0 1862.64    18.91853.787      27 1849.59    49.2 1839.73    52.1 1837.48
    78.8 1812.84    83.1 1811.84     108 1815.83  117.791816.764   124.1 1816.82
   132.1 1814.41  147.751805.509   156.3 1802.84   164.3 1802.32   176.4  1802.9
  183.31 1805.51   188.4 1806.95   196.5 1807.74   232.7 1809.03   236.7 1810.39
   248.7 1816.64   284.8 1826.88   296.8 1829.58   307.5 1833.25   344.8 1847.51
   352.8 1852.13   380.8 1866.09   392.8 1871.31   420.8 1886.38   429.9 1891.87
#Mann= 5 ,-1 , 0
       0      .1       0    18.9     .06       0  117.79      .1       0
  147.75    .045       0  183.31      .1       0
Bank Sta=147.75,183.31
XS Rating Curve= 0 ,0
Exp/Cntr(USF)=0,0
Exp/Cntr=0.3,0.1

Type RM Length L Ch R = 1 ,8349    ,251.9,254.2,255.6
XS GIS Cut Line= 4
2454557.27778638613767.9240534122454562.16434655613903.118884661
 2454554.0200796614035.0560091322454540.98925249614219.116442037
#Sta/Elev= 30
       0 1871.67      47 1851.28      55 1847.16   63.721843.741      95 1831.39
     103 1827.61     115    1816     123 1809.92     127 1807.83   131.1 1807.47
   155.1 1810.99  162.38 1811.23   167.1  1809.7   175.1 1803.88   178.11802.583
   187.2 1800.27   203.2 1799.62   211.2 1799.94   215.2 1800.91  218.931802.585
   223.2 1803.67   251.3 1805.01   295.4 1805.03   299.4  1805.6   327.5 1815.14
   355.5 1828.58   363.5 1833.02   375.6 1838.49  425.641869.353     452 1886.35
#Mann= 6 ,-1 , 0
       0      .1       0   63.72     .06       0  162.38      .1       0
   178.1    .045       0  218.93      .1       0  425.64      .1       0
Bank Sta=178.1,218.93
XS Rating Curve= 0 ,0
Exp/Cntr(USF)=0,0
Exp/Cntr=0.3,0.1

Type RM Length L Ch R = 1 ,8095    ,196,196.7,197.9
XS GIS Cut Line= 4
2454350.41340603613629.4715153862454317.83633826613865.655256724
2454296.66124421 614004.107794752454273.85729677614119.756385336
#Sta/Elev= 30
       0 1879.92    25.7  1868.7    90.3 1835.75    94.3 1833.24   106.4 1821.87
   122.6 1808.46   130.6 1803.93  140.211802.329   215.4 1800.33   259.8 1802.38
     268 1800.78  279.781796.166   284.2 1793.88   292.3 1792.84   308.5 1793.21
  317.091796.165  332.371799.681   340.8 1802.35   344.9 1804.49     357 1814.04
   377.3 1826.34     405  1845.6     418 1855.33   438.4 1871.91   450.7 1883.27
   458.8 1892.55   467.6 1899.98     471 1901.91   474.4 1902.81   496.4 1904.53
#Mann= 5 ,-1 , 0
       0      .1       0  140.21     .06       0  279.78    .045       0
  317.09     .06       0  332.37      .1       0
Bank Sta=279.78,317.09
XS Rating Curve= 0 ,0
Exp/Cntr(USF)=0,0
Exp/Cntr=0.5,0.3

Type RM Length L Ch R = 1 ,7898    ,56.5,57.1,58.1
XS GIS Cut Line= 4
2454182.64150702613596.8944476162454127.26049181613831.449335565
2454104.45654437613943.840219374 2454084.9103037614101.838998062
#Sta/Elev= 30
       0 1916.78    22.6 1905.54    98.71859.213  102.241856.915   125.4  1841.9
   133.6 1834.86   154.1  1820.2   178.8 1803.75   195.2 1797.64  207.511796.955
   215.8  1795.3   256.8 1798.06   261.3 1796.68  267.151791.865   273.1 1789.34
   289.4 1788.87   297.6 1789.63  302.611791.864  311.911795.653   338.4 1798.75
  371.311800.438     395  1803.3   414.41809.283   424.5 1812.44   438.9 1811.76
   451.5 1809.36   467.6 1812.13   487.7 1821.61   495.2 1824.03   514.9 1822.91
#Mann= 9 ,-1 , 0
       0      .1       0    98.7      .1       0  102.24      .1       0
  207.51    .035       0  267.15    .045       0  302.61    .035       0
  311.91      .1       0  371.31     .06       0   414.4    .055       0
#XS Ineff= 2 , 0
             250  1797.3     318          1797.3
Permanent Ineff=
       F       F
Bank Sta=267.15,302.61
XS Rating Curve= 0 ,0
Exp/Cntr(USF)=0,0
Exp/Cntr=0.5,0.3

Type RM Length L Ch R = 1 ,7841    ,116,115.5,115.7
XS GIS Cut Line= 4
 2454084.9103037613622.9561018322454081.65259693613785.841440686
2454044.18896899613935.6959524322454019.75616816614088.808170954
#Sta/Elev= 30
       0 1954.15    13.8 1951.18    19.9 1949.12    43.9 1935.97    50.8 1930.08
      57 1923.36    67.9 1909.45   85.251890.967   127.6  1839.5     132 1834.84
   172.2 1797.86   176.4 1795.54  181.041795.129  185.751795.646   209.4 1796.93
   213.5 1795.92  219.871790.871   221.7 1789.31   225.8 1787.98   250.6 1787.76
   255.2 1788.09  260.371790.872   265.1    1794   268.4 1794.95   295.9 1795.63
   316.6 1794.63   340.9 1794.89  394.911799.323  462.491807.961   472.4 1809.11
#Mann= 8 ,-1 , 0
       0      .1       0   85.25      .1       0  181.04    .055       0
  185.75     .06       0  219.87    .045       0  260.37     .06       0
  394.91    .055       0  462.49     .05       0
#XS Ineff= 2 , 0
          207.66 1797.01
Permanent Ineff=
       F       F
Bank Sta=219.87,260.37
XS Rating Curve= 0 ,0
Exp/Cntr(USF)=0,0
Exp/Cntr=0.5,0.3

Type RM Length L Ch R = 1 ,7725    ,166.7,161.5,156.2
XS GIS Cut Line= 4
2454016.49846138613609.9252747242453972.51941989 613736.97583903
 2453928.5403784613935.6959524322453939.94235212614150.704599719
#Sta/Elev= 30
       0 1944.89    17.9 1928.04      43  1895.4    66.5 1869.38      73  1863.9
    90.2 1852.17   102.8 1840.59   106.8 1835.24   115.3 1821.95  121.481816.389
   142.7 1802.86  152.211794.758   156.9 1792.06     161 1791.75   185.6 1794.12
   197.9 1794.04     202 1792.23  207.471788.017   210.2 1786.19   214.2 1785.29
   222.4 1785.06   234.7 1785.28  240.731788.022   242.9 1789.78   248.2 1791.73
   271.7 1792.31   305.3 1791.47   461.7 1794.49   521.4 1798.55   553.3 1799.51
#Mann= 5 ,-1 , 0
       0      .1       0  121.48    .055       0  152.21     .06       0
  207.47    .045       0  240.73     .05       0
#XS Ineff= 2 , 0
          190.32 1794.64  272.08          1792.4
Permanent Ineff=
       F       F
Bank Sta=207.47,240.73
XS Rating Curve= 0 ,0
Exp/Cntr(USF)=0,0
Exp/Cntr=0.3,0.1

Type RM Length L Ch R = 1 ,7564    ,186,192.9,199.2
XS GIS Cut Line= 4
2453834.06688187613556.173112902 2453801.4898141613712.543038202
2453808.00522765613826.1028068452453928.67716971614149.622911559
#Sta/Elev= 30
       01865.824  43.6351837.124  59.9781827.058  92.6661809.056 106.5481802.066
 121.2671790.465 125.3531788.559 130.218 1788.13 153.8881789.995 178.1051790.487
 186.1191789.357  192.951784.086 194.1321783.015 198.1381781.221 206.1511780.577
 222.1781780.993 226.1841782.229   228.51783.706 238.2041790.141 242.2111791.125
  266.251788.569 312.7381788.389 351.1611789.016 381.0451791.322 398.1221793.349
 430.1071792.499 534.2961795.204 577.4281795.352 607.3121796.648 618.766 1797.72
#Mann= 5 ,-1 , 0
       0    .035       0 106.548      .1       0  192.95    .045       0
   228.5      .1       0 381.045     .05       0
#XS Ineff= 2 , 0
             175 1790.52  244.62         1790.52
Permanent Ineff=
       F       F
Bank Sta=192.95,228.5
XS Rating Curve= 0 ,0
Exp/Cntr(USF)=0,0
Exp/Cntr=0.3,0.1

Type RM Length L Ch R = 1 ,7371    ,309.7,307,304.8
XS GIS Cut Line= 5
2453679.32580996613484.503563807 2453645.1198888613626.213808609
2453609.28511425613740.2335458072453822.34108119613909.882921086
2453910.79608506614147.223229814
#Sta/Elev= 30
       01848.442   23.031833.289  42.2371827.937  64.1791815.953  70.6651810.649
  88.8681791.769  98.5881784.715 108.5321783.552  135.051785.816 200.998 1785.94
  205.191785.477  212.131781.558   218.41778.272 230.3481777.689 234.5411777.923
   240.71781.285 247.1191785.594 275.9861787.107 301.6721785.258   340.21786.839
 365.886 1785.74 397.9931787.456 441.0131786.575 507.1581788.041 537.6471790.241
 555.7981794.248 585.3911794.188 616.4891795.837 653.8071793.626 790.9351796.126
#Mann= 4 ,-1 , 0
       0      .1       0  212.13    .045       0   240.7      .1       0
 653.807     .05       0
#XS Ineff= 2 , 0
                          358.06         1789.39
Permanent Ineff=
       F       F
Bank Sta=212.13,240.7
XS Rating Curve= 0 ,0
Exp/Cntr(USF)=0,0
Exp/Cntr=0.3,0.1

Type RM Length L Ch R = 1 ,7064    ,187.2,193.6,199.3
XS GIS Cut Line= 4
2453412.19385424613264.6083563542453322.60691787613660.419729769
2453306.31838398613785.8414406862453229.76227472614121.385238725
#Sta/Elev= 30
       0 1816.42    22.8 1801.99    51.6 1779.21    59.8 1775.52   68.571774.516
   158.2 1779.16   199.2 1777.75  267.471781.351   297.6 1778.59   314.1 1780.31
   334.5 1777.61  372.361778.468   387.9 1778.56   408.3 1781.61   416.4 1780.38
   425.8 1776.83   432.5 1773.79   444.6 1772.69   456.7 1773.17   465.31776.554
   472.9 1779.76   566.2 1781.75   603.1 1785.11   660.6 1786.64   689.3 1789.57
   733.3 1802.88   776.7 1819.97   791.9 1828.08   818.1 1844.66   876.5 1872.45
#Mann= 6 ,-1 , 0
       0      .1       0   68.57     .06       0  267.47     .05       0
  372.36      .1       0   425.8    .045       0   465.3      .1       0
#XS Ineff= 2 , 0
          266.13 1781.14
Permanent Ineff=
       F       F
Bank Sta=425.8,465.3
XS Rating Curve= 0 ,0
Exp/Cntr(USF)=0,0
Exp/Cntr=0.3,0.1

Type RM Length L Ch R = 1 ,6870    ,210.9,213.6,217.1
XS GIS Cut Line= 4
2453299.80297043613121.2692581632453145.06189852613624.584955221
2453081.53661636613800.501121183 2452977.2899995614031.798302355
#Sta/Elev= 30
       0  1823.4   19.441818.257    64.5 1799.65    75.8  1791.3   83.42 1781.84
    89.6 1774.74    97.9 1771.52  127.88 1773.64     175 1773.25   216.6 1776.52
   248.6 1774.12  307.581773.785   386.7 1773.05   457.8  1774.6   499.7 1776.31
   520.5 1779.12  531.281776.175   537.5 1774.28   558.3 1771.02   588.6 1771.33
   599.8 1774.19   609.8 1777.96   680.2 1782.61   703.4 1786.54   711.9 1789.48
   742.5 1804.96   808.6 1841.61   869.8 1872.35   922.4 1901.58   967.3 1923.31
#Mann= 8 ,-1 , 0
       0      .1       0   19.44      .1       0   83.42      .1       0
  127.88     .06       0  307.58     .05       0  531.28      .1       0
   537.5    .045       0   599.8      .1       0
#XS Ineff= 2 , 0
          216.34 1776.62
Permanent Ineff=
       F       F
Bank Sta=537.5,599.8
XS Rating Curve= 0 ,0
Exp/Cntr(USF)=0,0
Exp/Cntr=0.3,0.1

Type RM Length L Ch R = 1 ,6657    ,231.7,237.5,245.1
XS GIS Cut Line= 4
2453200.44291373613049.5997090672452978.91885289613494.276684138
2452881.18764957613683.2236772082452762.28135221 613881.94379061
#Sta/Elev= 30
       0 1819.41      50 1806.07    67.9 1804.39   85.131796.162   102.5  1787.9
   108.7 1783.48   121.5 1771.23   126.9 1769.75   184.7 1770.61     207 1773.02
  255.37 1771.77   309.8 1769.93   425.6 1770.21   488.4 1773.71   538.9 1774.47
     556 1777.26   569.5  1774.4     574 1771.05   578.6 1767.06   586.4 1766.14
   596.6 1766.79  613.941770.988     631 1776.66   641.6 1781.88   657.7 1783.59
   663.6 1785.51   677.6 1794.03   734.4 1822.47   830.3 1874.59   941.1 1928.28
#Mann= 7 ,-1 , 0
       0      .1       0   85.13      .1       0   126.9     .06       0
  255.37     .05       0   425.6      .1       0     574    .045       0
  613.94      .1       0
#XS Ineff= 1 ,-1
   85.22  210.77 1773.35
Permanent Ineff=
       F
Bank Sta=574,613.94
XS Rating Curve= 0 ,0
Exp/Cntr(USF)=0,0
Exp/Cntr=0.3,0.1

Type RM Length L Ch R = 1 ,6419    ,196.5,194.5,190.8
XS GIS Cut Line= 4
2453136.67631996612995.9480937512452861.17889499613327.751561786
2452706.33727657613472.5385296562452571.60495925613631.402008291
#Sta/Elev= 30
       0 1818.62    24.6 1812.24    45.4 1809.88    71.6  1804.9  103.931796.767
  125.551790.812     137 1783.99   149.4 1773.37   159.7 1769.32   197.1  1767.1
   206.6 1769.43   215.9 1769.89  257.321767.727   378.7 1766.82   435.9 1767.75
   500.3 1766.59  512.591768.668   517.3 1769.59   531.4 1769.01  538.84 1766.53
   544.1  1763.4   555.1  1762.6   573.9 1764.32  580.421766.526   587.9 1771.56
   593.4 1773.41   656.8 1782.63   673.5 1790.79   772.2 1827.99   851.6 1865.44
#Mann= 7 ,-1 , 0
       0      .1       0  103.93      .1       0  125.55    .055       0
  257.32     .05       0  512.59      .1       0  538.84    .045       0
  580.42      .1       0
#XS Ineff= 1 ,-1
  118.71  214.05 1769.94
Permanent Ineff=
       F
Bank Sta=538.84,580.42
XS Rating Curve= 0 ,0
Exp/Cntr(USF)=0,0
Exp/Cntr=0.3,0.1

Type RM Length L Ch R = 1 ,6225    ,342.6,339.8,336
XS GIS Cut Line= 4
2452977.81284133 612825.019034462452666.11867438613239.270636977
2452543.45193772613390.0903951752452444.91636236613494.658760859
#Sta/Elev= 30
       0  1834.5    22.4 1828.75   89.391803.436   117.5 1795.24   142.5 1794.25
   192.6 1778.59   212.1 1774.96   222.6 1768.43  227.071767.288  236.021765.411
   246.3 1764.18   277.9 1765.97     332 1763.13  364.74 1763.29   479.2 1763.15
  515.751766.867   543.7 1767.91   555.5 1764.52   561.8 1761.32     585 1760.52
   600.2 1761.49   608.7 1764.22   637.1 1765.65   703.5 1778.36   713.9  1783.1
   730.4 1787.07     743 1795.93   766.3 1806.23  815.44 1820.53   856.5  1839.4
#Mann= 9 ,-1 , 0
       0      .1       0   89.39      .1       0  227.07     .06       0
  236.02    .035       0  364.74     .05       0  515.75      .1       0
   555.5    .045       0   608.7      .1       0  815.44      .1       0
#XS Ineff= 2 , 0
          269.23 1768.31
Permanent Ineff=
       F       F
Bank Sta=555.5,608.7
XS Rating Curve= 0 ,0
Exp/Cntr(USF)=0,0
Exp/Cntr=0.3,0.1

Type RM Length L Ch R = 1 ,5885    ,261.9,266.4,269.4
XS GIS Cut Line= 4
2452706.33727657612601.8057923272452428.82892149612967.795072221
2452296.10753427613180.9536638072452207.62660946613307.642260693
#Sta/Elev= 30
       0 1835.33   42.64 1818.75    66.1  1808.9    96.7  1798.2     109 1795.76
   117.5 1791.54   138.4 1783.62   158.2  1773.6  193.221765.776   212.2 1763.77
   244.3 1762.33  317.011761.971   387.9 1763.56   454.21762.932   510.1 1762.23
   576.3 1759.76  585.181758.451   599.5 1754.07     607    1754   623.2 1754.73
  636.261758.451   657.6 1760.13   701.2 1767.87   726.8 1774.35     742 1781.83
  753.211783.609   756.7 1784.73   771.3 1793.97   836.3 1820.47   864.9 1833.58
#Mann= 8 ,-1 , 0
       0      .1       0   42.64      .1       0  193.22    .055       0
  317.01    .035       0   454.2      .1       0  585.18    .045       0
  636.26      .1       0  753.21      .1       0
#XS Ineff= 1 ,-1
  111.56  391.13  1763.7
Permanent Ineff=
       F
Bank Sta=585.18,636.26
XS Rating Curve= 0 ,0
Exp/Cntr(USF)=0,0
Exp/Cntr=0.3,0.1

Type RM Length L Ch R = 1 ,5618    ,91.4,83.2,76.9
XS GIS Cut Line= 4
2452565.57216892612489.1937062062452316.21683536612730.505319322
2452095.01452334612985.8934432042452050.77406094  613114.5929702
#Sta/Elev= 30
       0 1824.11    20.6 1816.97    70.7 1804.32      93 1802.75  124.871796.805
   132.31794.844   181.4 1777.49   192.7 1775.32   235.2 1773.13  293.941761.035
  376.251758.645  450.521756.844   538.3 1755.16   569.2  1756.7  578.381754.444
   587.5 1751.14   599.7 1750.44   609.2 1750.91  621.111754.445  635.141755.984
   648.9 1756.92   685.9 1763.75   702.8 1768.14   720.5 1775.58  734.131779.308
   740.9 1781.68   749.4 1782.53   770.5 1791.18  814.39 1803.74     821 1805.37
#Mann= 11 ,-1 , 0
       0      .1       0  124.87      .1       0   132.3    .055       0
  293.94     .02       0  376.25    .055       0  450.52      .1       0
  578.38    .045       0  621.11      .1       0  635.14     .05       0
  734.13      .1       0  814.39     .05       0
Bank Sta=578.38,621.11
XS Rating Curve= 0 ,0
Exp/Cntr(USF)=0,0
Exp/Cntr=0.5,0.3

Type RM Length L Ch R = 1 ,5535    ,62.1,64.1,67.3
XS GIS Cut Line= 4
2452408.99594399612348.0191710162452201.28803205612650.234182892
2452075.62474532612918.1773892982452040.31440029613096.806193569
#Sta/Elev= 30
       0 1820.91    27.8  1815.3    41.1 1811.07    61.7    1801      86 1791.82
   158.8 1784.32   202.2 1775.55   221.9 1773.26   270.4 1767.12   307.6 1759.17
     319 1757.77   348.9 1758.06   393.2 1755.87   508.8 1753.39   539.7 1754.89
     553 1752.84   570.7 1749.37   594.7 1749.71   604.1 1752.99   609.7 1756.04
   617.6 1757.43   645.7 1757.69   692.9 1762.64   708.3 1763.16   716.4 1765.42
   753.9 1770.86   769.4 1773.86   789.8 1781.96     802  1784.1   844.7 1799.55
#Mann= 6 ,-1 , 0
       0      .1       0    27.8     .05       0   221.9     .06       0
     553    .045       0   604.1     .06       0   753.9     .05       0
#XS Ineff= 2 , 0
             535 1754.28     619         1754.28
Permanent Ineff=
       F       F
Bank Sta=553,604.1
XS Rating Curve= 0 ,0
Exp/Cntr(USF)=0,0
Exp/Cntr=0.5,0.3

Type RM Length L Ch R = 1 ,5471    ,235.9,238.5,241.1
XS GIS Cut Line= 4
2452344.36985689612320.2755770242452181.48451804612595.773001999
2452012.56638886612905.4562388322451936.15104471612999.969953969
#Sta/Elev= 30
       0 1813.15    12.3 1808.33   25.891801.587    50.3 1790.31    73.2 1785.69
   114.6 1783.68   142.4 1781.23   165.7 1778.18  227.031768.102   301.9 1756.79
   332.7 1757.38   373.7 1754.91   469.4 1753.88   496.7 1753.81     515 1755.08
   519.5 1754.57  524.631752.304   530.7 1749.04   537.7 1748.18   559.7 1749.35
  569.011752.301   576.4 1753.28   626.5 1753.93   666.4 1758.78   679.8 1762.42
   715.8 1777.07  729.63 1781.35     757 1789.68   777.5 1794.38   794.3 1796.96
#Mann= 6 ,-1 , 0
       0      .1       0   25.89     .05       0  227.03     .06       0
  524.63    .045       0  569.01     .06       0  729.63     .05       0
Bank Sta=524.63,569.01
XS Rating Curve= 0 ,0
Exp/Cntr(USF)=0,0
Exp/Cntr=0.5,0.3
